--- MOYERRN.prj (project) ---

Proj Title=MOYERRN
Current Plan=p01
Default Exp/Contr=0,0
English Units
Geom File=g01
Flow File=f01
Plan File=p01
BEGIN DESCRIPTION:
Stream Name: Moyer Run
Flood Zone: Approximate
Pendleton County, West Virginia
HEC-RAS Version: 5.0.7
Hydrology Method:
Regression
Model Notes:
NA
END DESCRIPTION:
DSS Export Rating Curves= 0
DSS Export Rating Curve Sorted= 0
DSS Export Volume Flow Curves= 0
DXF OffsetX= 0
DXF OffsetY= 0
DXF ScaleX= 0
DXF ScaleY= 0

--- MOYERRN.p01 (plan) ---

Plan Title=Floodplain
Program Version=4.00
Geom File=g01
Flow File=f01
K Sum by GR=0
Std Step Tol=0.01
Critical Tol=0.01
Num of Std Step Trials=20
Max Error Tol=0.3
Flow Tol Ratio=0.001
Split Flow NTrial=30
Split Flow Tol=0.02
Split Flow Ratio=0.02
Log Output Level=0
Friction Slope Method=1
Unsteady Friction Slope Method=2
Unsteady Bridges Friction Slope Method=1
Global Log Level=0
CheckData=False
Run HTab=0
Run UNet=0
Run PostProcess=0
UNET Theta=0
UNET Theta Warmup=0
UNET ZTol=0
UNET ZSATol=0
UNET MxIter=0
UNET MaxInSteps=0
UNET DtIC=0
UNET DtMin=0
UNET MaxCRTS=0
UNET WFStab=0
UNET SFStab=0
UNET WFX=0
UNET SFX=0
UNET DSS MLevel=0
UNET DZMax Abort=0
UNET Convert EG Bridges=0
UNET Use Existing IB Tables=0
UNET Froude Limit=0
UNET Froude Power=0
Write IC File=0
Echo Input=False
Echo Output=False
Write Detailed=0

--- MOYERRN.f01 (steady flow) ---

Flow Title=Flows
Program Version=5.07
Number of Profiles= 6
Profile Names=P100yr,P10yr,P25yr,P50yr,P500yr,P101yr
River Rch & RM=MOYERRN,Main            ,9836
     556     260     367     459     814     676
River Rch & RM=MOYERRN,Main            ,7999
     646     302     427     533     948     786
River Rch & RM=MOYERRN,Main            ,4037
     837     390     552     690    1232    1019
River Rch & RM=MOYERRN,Main            ,3493
     931     432     613     767    1371    1133
Boundary for River Rch & Prof#=MOYERRN,Main            , 1
Up Type= 0
Dn Type= 3
Dn Slope=0.05
Boundary for River Rch & Prof#=MOYERRN,Main            , 2
Up Type= 0
Dn Type= 3
Dn Slope=0.05
Boundary for River Rch & Prof#=MOYERRN,Main            , 3
Up Type= 0
Dn Type= 3
Dn Slope=0.05
Boundary for River Rch & Prof#=MOYERRN,Main            , 4
Up Type= 0
Dn Type= 3
Dn Slope=0.05
Boundary for River Rch & Prof#=MOYERRN,Main            , 5
Up Type= 0
Dn Type= 3
Dn Slope=0.05
Boundary for River Rch & Prof#=MOYERRN,Main            , 6
Up Type= 0
Dn Type= 3
Dn Slope=0.05
DSS Import GetInterval= 0
DSS Import GetPeak= 0
DSS Import FillOption= 0

--- MOYERRN.g01 (geometry) ---

Geom Title=Geometry
Program Version=5.07

River Reach=MOYERRN         ,Main
Reach XY= 30
     2412379.623575802.7090000212412765.38100001575763.621000022
2412875.65500003575693.0780000092412982.50700003575720.072999999
2413387.96300003575998.6570000052413422.36200002576151.989999995
2413666.34099999576267.292000011     2414336.044 576151.99500002
     2414404.458576042.272000015     2414681.523575951.369000003
2415055.69499999576094.910999998     2415143.873 576185.54900001
     2415410.329576172.7900000212415689.91700003576393.069000006
      2416037.34576445.9150000212416078.64800003576618.709999993
     2416324.662576864.415000007     2416448.655576834.677000016
2416772.69200003577008.0949999992417087.24000001 577068.47300002
2417203.31400001576965.5520000012417690.23100001576776.131999999
2417919.64900002576839.986000001      2418257.78      576598.603
2419086.68100002576305.419000015     2419469.495576268.658999994
2419727.03999999576349.4590000062419998.69299999576216.233999997
2420514.54200003576231.5160000032420776.77998433575933.011930853

Type RM Length L Ch R = 1 ,9836    ,140.1,140.1,140.1
XS GIS Cut Line= 2
2412614.70021407576179.7081328092412192.21421407 575442.63713281
#Sta/Elev= 30
       0 2639.82    20.7 2637.73    35.9 2624.87      47 2620.47    73.4 2613.58
    77.4 2609.32    85.1 2593.99    90.6 2584.71    95.8 2579.02  156.692540.727
   229.5 2496.42   275.6  2473.1     294  2462.3   317.1 2451.86   349.4 2433.13
   366.4 2426.41   396.3 2418.96   409.3  2413.6     428 2412.86   441.6 2408.37
   446.2 2408.21   450.8 2408.42     460 2412.03   469.2 2420.75   483.1 2429.76
   521.8 2448.21   561.4 2472.74   579.9 2482.42   773.5 2600.73   849.6 2644.73
#Mann= 4 ,-1 , 0
       0      .1       0  156.69      .1       0   441.6    .045       0
   450.8      .1       0
Bank Sta=441.6,450.8
XS Rating Curve= 0 ,0
Exp/Cntr=0.3,0.1

Type RM Length L Ch R = 1 ,9696    ,87.8,90.1,92
XS GIS Cut Line= 2
     2412643.369       576174.22     2412418.347      575365.241
#Sta/Elev= 30
       0 2634.83    14.2 2631.68    25.5 2627.16    54.7 2612.03    74.2 2607.53
    87.2 2602.67    88.9 2601.49    90.5 2598.23   105.5 2563.56   106.7 2562.23
  146.272537.849   176.1  2522.2   217.1 2496.16   225.9 2492.41   254.9 2473.77
   296.5 2450.96   330.8 2428.39   350.4 2418.13   383.6 2406.25   412.7 2406.42
   426.72401.815   436.9 2401.29   441.72401.662   450.1 2402.65   458.4 2406.46
   489.9 2431.04   632.9 2518.38   710.8 2572.56   782.2 2609.36   839.7 2642.01
#Mann= 4 ,-1 , 0
       0      .1       0  146.27      .1       0   426.7    .045       0
   441.7      .1       0
Bank Sta=426.7,441.7
XS Rating Curve= 0 ,0
Exp/Cntr=0.3,0.1

Type RM Length L Ch R = 1 ,9606    ,64.2,65,65.6
XS GIS Cut Line= 3
2412657.14643727576163.0961051422412611.84474156575717.629430658
2412497.33212185575376.608332395
#Sta/Elev= 30
       0 2630.98   19.212624.573   38.922614.891    54.8 2608.06      87 2598.63
      91 2595.18      95 2586.83   107.1 2556.58   111.1 2548.66  136.582537.722
   151.5 2531.45   180.7 2514.66   243.7 2473.86     300 2440.46   320.1 2426.54
   364.3  2401.5   376.4 2398.04   397.2 2397.43   415.1 2394.11   420.6 2393.89
   424.7 2394.13   428.7  2394.8   440.7  2404.6   469.3 2413.47   507.2 2432.92
   533.2 2448.43   601.9 2493.89   699.9 2564.28   765.3 2599.27   807.5 2623.96
#Mann= 6 ,-1 , 0
       0      .1       0   19.21      .1       0   38.92      .1       0
  136.58      .1       0   415.1    .045       0   424.7      .1       0
#XS Ineff= 2 , 0
          386.86 2405.65
Permanent Ineff=
       F       F
Bank Sta=415.1,424.7
XS Rating Curve= 0 ,0
Exp/Cntr(USF)=0,0
Exp/Cntr=0.3,0.1

Type RM Length L Ch R = 1 ,9541    ,68.8,70.4,71.2
XS GIS Cut Line= 3
     2412686.445      576169.4382412678.70738044575718.487869527
2412568.56941294575353.837945673
#Sta/Elev= 30
       0 2628.18    33.1 2623.24    40.9 2621.07    50.12615.807    60.9 2608.83
    72.9 2603.59   105.9 2596.34   115.7 2592.52   120.9 2586.67   136.9 2558.01
  148.552541.254   176.9 2525.11   220.9 2496.61   328.9 2424.46   360.9 2401.21
   372.9 2395.88   400.9 2393.39   412.9 2390.17   420.9 2389.41   428.12389.997
   432.9 2391.27   440.9 2399.39   448.9 2403.83   469.7 2405.29   482.3 2409.01
     536    2436   607.8 2484.36   653.5 2518.21   719.7 2562.01   831.9 2623.44
#Mann= 5 ,-1 , 0
       0      .1       0    50.1      .1       0  148.55      .1       0
   412.9    .045       0   428.1      .1       0
#XS Ineff= 2 , 0
          397.68 2396.66
Permanent Ineff=
       F       F
Bank Sta=412.9,428.1
XS Rating Curve= 0 ,0
Exp/Cntr=0.3,0.1

Type RM Length L Ch R = 1 ,9470    ,82.1,79.8,76
XS GIS Cut Line= 3
2412749.00820913576163.0961051422412746.49144825575708.820767603
2412616.87826331575353.957484539
#Sta/Elev= 30
       0 2606.04    18.5 2606.84   53.562603.373   63.272604.034   142.5 2579.62
  152.172572.494   166.5 2545.21   170.5 2540.55   182.5 2531.21   198.5 2515.01
  250.792478.302   330.5 2425.64   370.5 2392.19   397.3 2385.99   398.5 2385.76
   403.6 2386.07   414.5 2387.88   434.5 2386.35   455.1 2399.22   471.5 2402.85
   492.8 2403.41     530 2422.45   576.8 2450.44   607.8 2472.06     612 2476.39
   623.5 2494.99   629.8 2502.84   639.1 2506.57   731.3 2560.53   832.1 2615.85
#Mann= 7 ,-1 , 0
       0      .1       0   53.56      .1       0   63.27      .1       0
  152.17      .1       0  250.79      .1       0   397.3    .045       0
   403.6      .1       0
Bank Sta=397.3,403.6
XS Rating Curve= 0 ,0
Exp/Cntr(USF)=0,0
Exp/Cntr=0.3,0.1

Type RM Length L Ch R = 1 ,9390    ,76.5,80.4,84.6
XS GIS Cut Line= 3
     2412820.744       576163.852412831.24256094575765.925295324
2412657.39987811575337.773668283
#Sta/Elev= 30
       0 2578.22    51.8 2577.52   107.3 2581.69   143.3 2577.59  164.942571.151
   171.3 2568.21   183.3 2551.11   199.3 2541.09   215.3 2509.18  264.072473.434
   307.3 2443.75   383.4  2395.6   395.4 2385.42   425.4 2382.88   433.32380.025
   438.3 2379.68   441.1 2379.94   452.5 2383.28   468.5 2393.53   480.1 2398.04
     516  2401.8   567.8 2430.08   619.6  2461.8   623.9  2469.7   636.7  2498.8
   641.2 2503.25   667.1 2514.37   762.1 2563.77   790.2 2581.25   860.2 2619.04
#Mann= 5 ,-1 , 0
       0      .1       0  164.94      .1       0  264.07      .1       0
   433.3    .045       0   441.1      .1       0
#XS Ineff= 2 , 0
          412.01 2391.89
Permanent Ineff=
       F       F
Bank Sta=433.3,441.1
XS Rating Curve= 0 ,0
Exp/Cntr=0.3,0.1

Type RM Length L Ch R = 1 ,9310    ,101.9,102.8,104.1
XS GIS Cut Line= 3
2412852.19540491576155.5458225242412888.68843757575648.418506656
2412798.08504615575340.115299739
#Sta/Elev= 30
       0 2558.63      34 2562.64    79.2  2561.7    87.2 2562.55    95.2 2565.79
   107.2 2568.11   139.3 2565.92  163.022555.673   199.5 2539.22   203.5 2531.44
   211.5 2509.56   215.5 2501.38   263.12466.708   307.7 2437.36   383.9 2392.18
   391.9 2384.97     408  2383.6     420  2377.9   444.1 2379.49   460.5 2373.88
   464.1 2373.41   468.3 2373.75   488.2 2383.34   545.7 2418.66   587.4 2450.07
   655.7 2491.78   720.2 2525.93   770.8 2555.57   820.9 2581.72   829.8 2587.38
#Mann= 5 ,-1 , 0
       0      .1       0  163.02      .1       0   263.1      .1       0
   460.5    .045       0   468.3      .1       0
#XS Ineff= 2 , 0
          440.91 2382.15
Permanent Ineff=
       F       F
Bank Sta=460.5,468.3
XS Rating Curve= 0 ,0
Exp/Cntr(USF)=0,0
Exp/Cntr=0.3,0.1

Type RM Length L Ch R = 1 ,9207    ,96.8,102.4,107.2
XS GIS Cut Line= 3
2412891.62967798576167.7621121892412992.13257064575675.711097642
2412945.56618074575333.546224377
#Sta/Elev= 30
       0 2542.36    23.7 2534.27    76.7 2530.79    93.1  2531.5   117.6 2536.51
   166.5 2541.57  188.822536.286   211.4 2526.63   215.5 2523.36   244.1 2487.45
   272.7 2464.16  292.862450.036   346.7 2414.98   395.1 2387.62   407.4 2378.31
   427.8 2377.32   441.6  2369.2   451.8 2367.57   456.4 2367.24   460.5 2367.46
   472.7 2371.29   489.5 2371.43   493.1  2372.8   505.3 2382.94   525.5 2390.45
   573.9 2421.62   618.3 2447.51   723.3 2501.05   769.2 2529.45   847.5  2581.3
#Mann= 5 ,-1 , 0
       0      .1       0  188.82      .1       0  292.86      .1       0
   451.8    .045       0   460.5      .1       0
Bank Sta=451.8,460.5
XS Rating Curve= 0 ,0
Exp/Cntr=0.3,0.1

Type RM Length L Ch R = 1 ,9105    ,83.5,81.1,78.9
XS GIS Cut Line= 4
2412910.07067641576164.6542620132413046.78361272575794.907911559
2413096.71947304 575740.726865992413193.04220355575387.543520803
#Sta/Elev= 30
       0 2537.37    34.2 2521.93    51.3 2517.41    89.6 2511.25     111 2511.74
     128 2515.51   171.6 2519.34   204.8 2515.62   213.3 2508.28   230.4 2484.61
   234.6 2480.33     283 2440.03   302.8 2426.04   332.8 2407.89   404.2 2366.85
   413.6  2364.9   420.82365.144   430.32365.558   451.4 2365.66   462.6 2369.74
   530.6 2385.82   575.8 2405.16   588.2 2415.37   613.1 2427.55   662.8 2443.58
   706.5 2464.37   745.8 2487.91   766.5 2503.93   778.9 2511.44     834 2535.52
#Mann= 3 , 0 , 0
       0      .1       0   420.8    .045       0   430.3      .1       0
Bank Sta=420.8,430.3
XS Rating Curve= 0 ,0
Exp/Cntr(USF)=0,0
Exp/Cntr=0.3,0.1

Type RM Length L Ch R = 1 ,9024    ,131.5,134.2,135.1
XS GIS Cut Line= 2
2412936.46790236576182.8751121892413337.66979017575441.590780471
#Sta/Elev= 30
       0  2545.1    52.6 2514.63    79.9 2500.89   102.7  2491.6   148.1 2477.61
   170.7 2472.78   211.8 2466.61   243.6 2454.16   275.5 2436.98   327.1 2404.13
   374.3 2380.13   398.3 2360.82   402.8  2358.9   415.6 2359.34   423.12357.063
   430.1 2356.63   433.3 2357.08   436.3 2358.14   445.1 2364.75   475.6 2367.77
   523.3 2382.51   556.9 2395.48   589.7 2413.08   690.1 2451.86   716.6 2464.01
   775.7 2488.64   793.9 2493.95   812.1 2496.65   825.8 2499.99   842.9 2505.87
#Mann= 3 ,-1 , 0
       0      .1       0   423.1    .045       0   433.3      .1       0
Bank Sta=423.1,433.3
XS Rating Curve= 0 ,0
Exp/Cntr=0.3,0.1

Type RM Length L Ch R = 1 ,8890    ,242.8,246.4,250.3
XS GIS Cut Line= 3
2412997.22743549576209.8240552092413357.65244937575718.900329406
2413551.84696116575589.955173578
#Sta/Elev= 30
       0 2552.87    55.5 2522.42    95.2    2497   175.7 2449.37   223.6 2427.35
   311.5 2391.47     329 2382.03   345.3 2368.55   358.8  2352.1   365.5 2349.27
   368.7 2349.08   373.7 2349.29   393.1 2351.55   403.5 2355.72   414.8 2357.11
   428.3 2357.42   450.4 2354.11   472.9 2356.87   497.7 2362.13   510.4 2366.99
   513.3 2368.49   516.2 2372.75   522.5 2387.38   527.7 2396.55   573.4 2427.47
     597 2446.66   699.9 2506.66  754.412526.806   795.2 2539.53   842.1 2550.22
#Mann= 4 ,-1 , 0
       0      .1       0   365.5    .045       0   373.7      .1       0
  754.41      .1       0
#XS Ineff= 2 , 0
                          421.65            2360
Permanent Ineff=
       F       F
Bank Sta=365.5,373.7
XS Rating Curve= 0 ,0
Exp/Cntr(USF)=0,0
Exp/Cntr=0.3,0.1

Type RM Length L Ch R = 1 ,8643    ,192.9,187.7,184
XS GIS Cut Line= 3
2413067.13745974576240.8951770962413457.08003941 576015.62954342
2413674.57789261575754.632119576
#Sta/Elev= 30
       0 2548.27    34.2 2532.76    44.4 2526.29    58.2 2519.58    67.5 2513.99
    76.7 2506.38   164.5 2453.11   186.5 2442.26   210.7 2432.31   235.5    2418
   312.4 2369.48   353.9 2339.88   359.2 2337.55   386.2 2338.46   394.3 2336.63
     400 2336.21   403.1 2336.53   411.9 2338.33   420.7    2343   432.4 2344.09
     450 2349.64   490.7 2372.92   519.8 2385.71  558.66 2408.93   607.2 2437.36
  622.082445.075   643.1 2456.59  690.232480.016   716.9 2491.59   790.1 2517.45
#Mann= 6 ,-1 , 0
       0      .1       0   394.3    .045       0   403.1      .1       0
  558.66      .1       0  622.08      .1       0  690.23      .1       0
Bank Sta=394.3,403.1
XS Rating Curve= 0 ,0
Exp/Cntr(USF)=0,0
Exp/Cntr=0.3,0.1

Type RM Length L Ch R = 1 ,8455    ,175.8,173.7,172
XS GIS Cut Line= 2
2413316.12838833576490.7108330022413705.47639715575784.897693857
#Sta/Elev= 30
       0 2486.62    20.7 2471.58    89.3 2436.18   110.6 2425.63   153.2  2409.5
   185.2  2395.6     240 2368.14   270.5 2348.71   285.2 2341.67   331.4 2326.93
     359 2326.83   363.3 2326.56   365.92326.886   386.2 2333.04     403 2333.55
     417 2336.23   435.4 2343.81   450.2 2350.91   468.4 2362.54   473.7 2367.95
  481.342380.467   488.4 2390.18   495.8 2397.09   516.3 2407.21   526.6  2417.1
   532.3 2420.63   550.6 2427.33     578  2433.9   687.6 2477.39   806.1 2514.52
#Mann= 4 ,-1 , 0
       0      .1       0     359    .045       0   365.9      .1       0
  481.34      .1       0
Bank Sta=359,365.9
XS Rating Curve= 0 ,0
Exp/Cntr(USF)=0,0
Exp/Cntr=0.3,0.1

Type RM Length L Ch R = 1 ,8282    ,153.7,149.1,145.6
XS GIS Cut Line= 2
2413550.12078772576584.6913868562413766.85145273575804.077398725
#Sta/Elev= 30
       0 2496.66    29.2 2481.62    74.4  2462.7   141.3 2427.23   162.1 2421.01
   178.7 2422.17     187 2410.89   199.4 2383.07   204.3 2375.83   281.8 2327.88
   315.6 2320.91     331  2313.5   332.2 2313.38   337.5 2313.52     353 2318.78
   377.9 2318.52   394.5 2326.65   398.6 2330.65   411.1 2353.11  436.322365.128
   444.7 2369.65   477.5 2378.99   481.7 2381.84   496.7    2401     526 2410.96
   564.7 2432.67   584.4 2447.02   734.9 2497.34     793 2511.94   810.1 2513.46
#Mann= 4 ,-1 , 0
       0      .1       0     331    .045       0   337.5      .1       0
  436.32      .1       0
#XS Ineff= 2 , 0
                          354.47         2319.29
Permanent Ineff=
       F       F
Bank Sta=331,337.5
XS Rating Curve= 0 ,0
Exp/Cntr(USF)=0,0
Exp/Cntr=0.3,0.1

Type RM Length L Ch R = 1 ,8133    ,135.1,133.6,133.9
XS GIS Cut Line= 3
 2413864.7561742576597.7949612222413778.35927565576220.276994363
2413778.35927565575811.749280673
#Sta/Elev= 30
       0 2441.88    33.8 2426.52    70.6 2417.44    98.4 2399.82   127.3 2387.13
   144.9 2382.91   214.7  2360.2   222.9 2355.97   230.8 2349.03   239.3 2343.75
   288.5 2320.12   296.7 2317.55   313.1 2315.55   333.6 2307.73   345.9 2306.58
   354.4  2303.8   358.3 2303.51   362.4 2303.67   366.5 2304.48   374.7 2311.23
   378.8 2313.01     391 2314.19   399.8 2320.09     439  2336.2  460.612347.264
     507 2370.36   598.1 2423.71     703 2475.91   766.9 2504.24   795.8 2510.01
#Mann= 4 ,-1 , 0
       0      .1       0   354.4    .045       0   362.4      .1       0
  460.61      .1       0
Bank Sta=354.4,362.4
XS Rating Curve= 0 ,0
Exp/Cntr(USF)=0,0
Exp/Cntr=0.3,0.1

Type RM Length L Ch R = 1 ,7999    ,126.3,125.6,125
XS GIS Cut Line= 3
2414003.43311228576555.9908764912413897.16987543 576160.30013927
2413788.11023761575813.546419019
#Sta/Elev= 30
       0  2446.4    65.7  2417.8   127.8 2392.57   169.2 2377.46   185.8  2372.9
   198.2  2367.6     281 2316.07   285.1 2314.36   314.2 2308.06   334.9 2306.35
     339 2304.94   351.4 2297.98   363.9 2297.77   376.3 2295.22   380.4 2295.02
   381.5 2295.24   384.6 2295.89   392.9 2301.61     406 2302.62   415.9 2305.67
  441.512320.388   480.7  2344.3   543.6  2378.3   564.6 2390.62   648.5 2440.76
   665.2 2452.04   707.1 2477.97   723.9 2486.42   744.1 2498.29   773.2 2507.55
#Mann= 4 ,-1 , 0
       0      .1       0   376.3    .045       0   381.5      .1       0
  441.51      .1       0
Bank Sta=376.3,381.5
XS Rating Curve= 0 ,0
Exp/Cntr(USF)=0,0
Exp/Cntr=0.3,0.1

Type RM Length L Ch R = 1 ,7874    ,134.7,138.5,142.9
XS GIS Cut Line= 3
2414075.60961115 576531.982379152414034.99860873576194.292606303
      2413907.57      575778.175
#Sta/Elev= 30
       0 2461.01    23.6 2457.43    55.8 2448.69   111.4 2429.59   164.6 2408.24
   180.7 2400.07     221 2376.71   253.1 2352.29   265.3 2344.63   309.6 2310.04
   325.7    2299   333.8 2295.21   354.5 2291.98   362.8 2287.83     367 2287.26
   372.7 2287.77   384.4 2290.08   392.1 2290.48   400.5 2293.64   412.8 2295.45
   421.4 2300.71   427.22302.947   461.2 2307.55     480 2314.02   544.5 2347.63
  624.272393.674     678 2424.32   693.3 2431.68   741.5 2457.99   775.3 2478.15
#Mann= 5 ,-1 , 0
       0      .1       0   362.8    .045       0   372.7      .1       0
   427.2      .1       0  624.27      .1       0
Bank Sta=362.8,372.7
XS Rating Curve= 0 ,0
Exp/Cntr=0.3,0.1

Type RM Length L Ch R = 1 ,7735    ,118.4,114.5,110.6
XS GIS Cut Line= 3
2414121.01301212 576526.918978182414161.70080436576141.822983029
2414005.65517382575778.730608728
#Sta/Elev= 30
       0 2465.93    22.5 2463.08    42.6 2459.41    58.7 2455.51    70.8 2451.36
    94.9 2440.67     159 2405.51   224.5 2365.76   259.8 2340.05   282.7 2323.06
     300 2309.14   312.5 2297.37   324.1 2282.77   328.2  2279.7   332.2 2278.46
   336.2 2278.26   340.2 2278.57   348.3 2281.67   360.3 2282.59   376.4 2288.85
   397.3 2288.99   427.8 2291.02  442.79 2290.76   484.4 2288.71   491.9 2288.96
     501 2290.89   572.4 2324.92  644.192363.178     712 2399.71   782.4    2442
#Mann= 5 ,-1 , 0
       0      .1       0   332.2    .045       0   340.2      .1       0
  442.79      .1       0  644.19      .1       0
Bank Sta=332.2,340.2
XS Rating Curve= 0 ,0
Exp/Cntr=0.3,0.1

Type RM Length L Ch R = 1 ,7621    ,208.7,206.9,204.7
XS GIS Cut Line= 3
2414249.50994909576555.0926014552414288.66601119576235.802965453
     2414122.546       575743.74
#Sta/Elev= 30
       0 2467.18    22.7 2458.18    71.1 2440.92    87.2 2434.33   156.6 2400.96
   228.2 2363.81   300.8 2329.71   316.9 2320.99   346.2 2302.18     371  2281.5
   375.8 2276.96     380 2274.06   389.9 2271.68   396.2 2271.22   398.2  2271.6
   401.1 2272.41   413.7 2280.94     418 2282.91   422.2 2283.89   439.1 2284.72
  490.312282.705   536.2 2284.04   578.4 2282.56   586.8 2283.71   595.3 2286.87
   619.4 2299.69   662.8 2325.44   699.2 2345.17   729.6 2362.48     841 2428.48
#Mann= 4 ,-1 , 0
       0      .1       0   389.9    .045       0   398.2      .1       0
  490.31      .1       0
Bank Sta=389.9,398.2
XS Rating Curve= 0 ,0
Exp/Cntr=0.3,0.1

Type RM Length L Ch R = 1 ,7414    ,148.9,151.7,153.9
XS GIS Cut Line= 3
2414390.06772436 576508.823818912414483.01587859576168.689342179
2414191.55801212575698.297990302
#Sta/Elev= 30
       0 2434.16    16.9 2430.64    33.5 2425.09    62.5 2411.49     104 2388.81
   182.7 2341.97     220 2322.41   240.9 2314.96   278.1 2304.26   352.6 2275.25
   366.9 2274.05   420.7 2273.76   432.3 2271.92   446.8    2268   475.1 2267.41
   487.5 2261.22   496.2 2260.73   503.3 2260.62   504.9 2260.75   510.7 2262.26
   522.1 2268.62   528.2 2270.55   559.8 2272.44   592.7 2272.37   620.9 2274.65
     635 2280.23  644.092285.199   696.6 2315.13   837.4 2391.92     906 2431.24
#Mann= 4 ,-1 , 0
       0      .1       0   496.2    .045       0   504.9      .1       0
  644.09      .1       0
Bank Sta=496.2,504.9
XS Rating Curve= 0 ,0
Exp/Cntr=0.3,0.1

Type RM Length L Ch R = 1 ,7262    ,108.3,111.4,112.7
XS GIS Cut Line= 3
2414598.00998303 576443.710801942414601.86291981576174.282144118
2414426.10721018575595.764591757
#Sta/Elev= 30
       0 2328.15    79.2 2310.88   131.2 2296.33     158 2290.19   266.7 2270.01
   300.5 2266.75   354.5 2264.14   412.3 2263.14   431.5 2263.99   434.3  2263.7
   450.7 2252.12   453.9 2250.94   459.3 2249.97   463.5 2250.86   463.5 2250.87
   471.9 2253.82   488.6 2254.29   505.3  2259.3   555.5 2262.64   563.8 2263.96
   593.1 2273.77  621.452286.765   639.1 2296.28   671.9  2311.3   697.6 2321.61
   714.3 2329.83   742.5 2341.19   793.7 2364.38  818.452373.616   874.1 2394.57
#Mann= 5 ,-1 , 0
       0      .1       0   453.9    .045       0   463.5      .1       0
  621.45      .1       0  818.45      .1       0
#XS Ineff= 2 , 0
          433.83 2271.89  498.88         2269.22
Permanent Ineff=
       F       F
Bank Sta=453.9,463.5
XS Rating Curve= 0 ,0
Exp/Cntr=0.3,0.1

Type RM Length L Ch R = 1 ,7151    ,114.9,123.7,128.5
XS GIS Cut Line= 3
2414628.42957964576436.5064033942414666.18014211576172.883943634
     2414617.947      575553.851
#Sta/Elev= 30
       0 2323.47    36.3 2313.82     101  2299.8   181.8 2284.21   298.7 2264.35
     338 2260.76   358.9 2259.83   431.1 2254.25   451.2  2249.1   467.2 2249.52
   471.2 2248.79   475.2 2246.86   482.22245.581   490.6 2245.44     492  2245.5
   511.3  2249.3   527.4 2249.38   559.5 2252.64   567.5 2256.64   594.8  2275.7
   603.6 2280.04   659.8 2300.27   695.9 2315.03  722.172326.959     740 2334.76
   760.1 2341.31   772.1 2343.01   804.2 2345.48  819.982347.732   887.2 2359.81
#Mann= 5 ,-1 , 0
       0      .1       0   482.2    .045       0     492      .1       0
  722.17      .1       0  819.98      .1       0
#XS Ineff= 2 , 0
          466.26 2251.29  517.42         2251.64
Permanent Ineff=
       F       F
Bank Sta=482.2,492
XS Rating Curve= 0 ,0
Exp/Cntr=0.3,0.1

Type RM Length L Ch R = 1 ,7027    ,104.1,102.7,102.2
XS GIS Cut Line= 4
2414668.31761969576434.9762201552414721.82899628576044.861023135
2414801.23297443575932.659749656 2414740.8169041 575632.30557142
#Sta/Elev= 30
       0 2323.06    38.8 2309.93    71.1 2301.98   131.6 2291.41   192.2 2277.93
   220.5 2273.57   248.1 2270.53   345.6 2256.06     390 2251.48   394.1 2250.53
   410.9 2243.62   423.5 2240.16   448.2  2240.7   460.92239.962   468.3  2239.6
   470.12239.613   476.9 2240.52   482.6 2242.58   492.1 2243.65   501.9 2246.38
   528.5 2247.78   547.6 2250.38   563.9 2256.32   574.12261.129   600.6 2271.63
     621 2277.76   694.2 2290.67  769.352308.187   804.6 2315.24   837.6 2319.84
#Mann= 5 ,-1 , 0
       0      .1       0   460.9    .045       0   470.1      .1       0
   574.1      .1       0  769.35      .1       0
Bank Sta=460.9,470.1
XS Rating Curve= 0 ,0
Exp/Cntr(USF)=0,0
Exp/Cntr=0.3,0.1

Type RM Length L Ch R = 1 ,6924    ,49.1,47,45.9
XS GIS Cut Line= 4
2414704.77675088576452.7267073352414763.31714943576189.179963581
2414891.67017833575962.5669719332414831.41969754575632.230492304
#Sta/Elev= 30
       0 2329.47    61.6 2305.77    97.9 2295.42   135.4 2286.23   161.6  2281.3
     246 2269.96   301.3 2260.12   367.2 2250.08     381 2245.76   394.8 2237.93
   398.1 2237.05   408.6 2236.73   420.3 2234.62   436.1  2235.5   445.3 2232.64
   449.9 2232.29   452.7 2232.52   459.1 2234.14   463.7 2237.12   468.3 2238.26
   491.3 2239.02   509.6 2238.24   530.4 2240.09     569 2249.93  616.712258.462
   735.7 2282.42   764.1  2285.7   829.8  2290.3     847 2293.33   866.2 2299.66
#Mann= 4 ,-1 , 0
       0      .1       0   445.3    .045       0   452.7      .1       0
  616.71     .05       0
#XS Ineff= 2 , 0
          435.98  2235.9
Permanent Ineff=
       F       F
Bank Sta=445.3,452.7
XS Rating Curve= 0 ,0
Exp/Cntr=0.5,0.3

Type RM Length L Ch R = 1 ,6877    ,38.5,38.3,38.2
XS GIS Cut Line= 3
 2414747.4324539576442.1727659572414926.55569299575964.685040252
2414863.61799474 575634.48395432
#Sta/Elev= 30
       0 2322.77    24.5 2313.23    99.1 2290.03   111.5 2284.78   121.3 2284.01
   142.7 2277.36   168.3 2271.13   202.5 2264.21   245.2 2257.12   262.3 2256.62
   309.3 2251.17   326.4 2247.44   347.7 2241.03   364.8 2237.95   372.4 2235.32
   394.7 2232.67   403.5 2229.98   409.7  2229.7   412.8 2229.87   433.2 2234.74
   488.7 2236.29   530.4 2240.49   575.2 2250.37  603.762253.847   660.7 2264.21
   697.4  2267.8   717.7  2270.8   795.1 2275.82   811.4 2280.33   846.1 2294.28
#Mann= 4 ,-1 , 0
       0      .1       0   403.5    .045       0   412.8      .1       0
  603.76     .05       0
#XS Ineff= 2 , 0
             380    2234     430            2234
Permanent Ineff=
       F       F
Bank Sta=403.5,412.8
XS Rating Curve= 0 ,0
Exp/Cntr(USF)=0,0
Exp/Cntr=0.5,0.3

Type RM Length L Ch R = 1 ,6839    ,87.5,81.6,76.9
XS GIS Cut Line= 3
2414778.19286457 576468.738575172414957.31610366575991.250849465
2414894.37840541575661.049763533
#Sta/Elev= 30
       0 2330.93    33.7 2318.47    81.4 2302.41     102 2294.86   111.4 2290.15
   124.1 2288.78   141.2 2281.93   179.6 2270.98   265.1 2251.43   290.7 2249.32
   307.8 2249.17   320.6 2247.78   412.7 2227.67   418.7 2227.23   425.1 2227.74
   444.5  2231.6   457.3 2231.96   471.7 2233.62  484.68 2233.51     509 2234.63
   545.3 2238.43   573.8 2239.78   606.3 2247.67   659.3 2253.81     704 2261.68
   768.7 2264.83   785.8 2266.31   826.2 2272.14   833.7 2274.39   846.1 2279.92
#Mann= 4 ,-1 , 0
       0      .1       0   412.7    .045       0   425.1      .1       0
  484.68     .05       0
#XS Ineff= 2 , 0
          399.25 2235.42  452.53         2235.38
Permanent Ineff=
       F       F
Bank Sta=412.7,425.1
XS Rating Curve= 0 ,0
Exp/Cntr=0.5,0.3

Type RM Length L Ch R = 1 ,6757    ,49.3,55.3,62.8
XS GIS Cut Line= 3
2414831.90747146576473.0771526412415010.59749342576130.797673942
2414937.61142811575660.163390729
#Sta/Elev= 30
       0 2327.84    72.6 2301.62    81.8 2296.99    90.8 2296.29     145 2278.93
     212 2260.44   284.8 2243.48   316.4 2237.36   348.9 2232.33   375.1 2226.04
   388.4 2224.36   408.6 2227.85   413.7 2226.88   424.8 2221.34   428.8 2221.03
   434.52221.454   441.7 2224.11   453.1 2226.76  461.83 2226.88   493.6 2231.53
   546.8 2236.55   602.9 2240.37   651.9 2247.86     722 2255.11   756.7  2257.7
   772.9 2256.53     789 2259.72   825.5 2262.97   837.6 2265.89   862.4 2276.38
#Mann= 4 ,-1 , 0
       0      .1       0   424.8    .045       0   434.5      .1       0
  461.83     .05       0
#XS Ineff= 2 , 0
          407.62 2227.79  458.32         2229.86
Permanent Ineff=
       F       F
Bank Sta=424.8,434.5
XS Rating Curve= 0 ,0
Exp/Cntr(USF)=0,0
Exp/Cntr=0.3,0.1

Type RM Length L Ch R = 1 ,6702    ,129.7,126.4,127.2
XS GIS Cut Line= 3
     2414852.285      576483.4582415105.21509437576006.498085933
2415015.83851902575658.802371877
#Sta/Elev= 30
       0 2328.11      35 2314.46    79.9 2299.32    91.7 2297.73   113.3 2290.19
   130.1 2285.76   202.5 2263.26   258.4 2248.44   315.7  2235.9   340.2 2231.27
     358 2226.31   366.8 2224.56   392.6 2221.57   434.9 2218.84   442.4 2218.47
     447 2218.91   465.1 2221.47   483.2 2230.48   499.22231.306   519.4 2229.93
   539.9 2229.89   620.3 2234.05   636.8 2236.14   665.7 2242.12   690.5 2246.06
   731.9 2249.82   814.4 2254.26   843.6 2257.81   872.2 2265.88   898.9 2274.84
#Mann= 4 ,-1 , 0
       0      .1       0   434.9    .045       0     447      .1       0
   499.2     .05       0
#XS Ineff= 2 , 0
          397.46 2224.93
Permanent Ineff=
       F       F
Bank Sta=434.9,447
XS Rating Curve= 0 ,0
Exp/Cntr=0.3,0.1

Type RM Length L Ch R = 1 ,6576    ,185.6,181.3,178.9
XS GIS Cut Line= 3
2415013.97794181576539.8695820592415193.30172491  576037.2584966
2415126.19514472575721.766188363
#Sta/Elev= 30
       0 2349.19    57.7 2334.52    71.5 2328.18    84.2 2327.94   109.7 2319.88
   152.2  2310.5   203.1 2292.17   258.8 2264.29   292.3 2245.64   326.3 2235.77
   347.5 2226.48     356 2221.89   369.92210.803     373 2209.86   380.8 2210.97
   385.7 2213.37   396.5 2213.22     409 2215.19   440.9 2216.53   457.9 2222.07
   468.5 2223.79  544.992222.621   562.9 2221.59   587.5 2225.07   640.6 2228.07
   652.9 2229.55   689.7 2237.34   719.6 2242.35   783.7 2250.53   856.2 2256.49
#Mann= 4 ,-1 , 0
       0      .1       0   369.9    .045       0   380.8      .1       0
  544.99     .05       0
#XS Ineff= 2 , 0
                          410.88         2215.72
Permanent Ineff=
       F       F
Bank Sta=369.9,380.8
XS Rating Curve= 0 ,0
Exp/Cntr=0.3,0.1

Type RM Length L Ch R = 1 ,6394    ,143.3,151.9,157.7
XS GIS Cut Line= 4
2415150.00297091576559.7907873932415318.38759903 576230.82002182
2415320.53796904 576097.381117452415245.62617139575747.329195636
#Sta/Elev= 30
       0 2338.31    35.1 2328.19   108.9 2301.44   182.9 2278.98     201 2268.23
   241.8 2248.95   273.2 2237.35   358.6 2213.01   367.5 2208.87   375.8 2202.79
   379.8 2201.05   387.8 2200.27   395.8 2202.34   411.8  2203.4   415.8 2202.94
   426.92197.982   431.8  2197.4     438 2197.87   443.8 2200.43   451.8 2206.64
   465.2 2211.82   475.8  2214.1  495.66 2214.58   573.8 2215.36   585.6 2216.79
   654.6 2219.51   745.1  2232.7   792.8 2237.79   847.4 2248.63     861 2250.34
#Mann= 4 ,-1 , 0
       0      .1       0   426.9    .045       0     438      .1       0
  495.66     .05       0
Bank Sta=426.9,438
XS Rating Curve= 0 ,0
Exp/Cntr=0.3,0.1

Type RM Length L Ch R = 1 ,6242    ,164.6,162.7,160.1
XS GIS Cut Line= 4
2415229.27778497 576603.868198062415421.53238885576246.219811637
 2415509.2950345 576154.707337332415458.08690302575823.645765573
#Sta/Elev= 30
       0 2313.34      38 2305.66    67.4 2298.52   144.6 2277.71   165.2  2270.9
   212.2 2251.95   235.8 2245.03   318.5 2225.68   376.1 2214.35   398.2 2205.95
   413.9 2197.28   419.4 2195.72   430.5 2194.83     4452191.517     452 2191.25
   453.52191.529   463.5  2194.7   477.8 2196.48   486.6 2200.14     497 2201.47
   506.1 2205.36   511.7 2206.21   571.4 2203.17  611.22 2203.46   636.2 2203.09
   680.7 2208.39   737.4 2209.98   777.8  2214.3   827.5  2217.7   867.8 2224.78
#Mann= 4 ,-1 , 0
       0      .1       0     445    .045       0   453.5      .1       0
  611.22     .05       0
Bank Sta=445,453.5
XS Rating Curve= 0 ,0
Exp/Cntr=0.3,0.1

Type RM Length L Ch R = 1 ,6080    ,77.2,77.6,77.6
XS GIS Cut Line= 3
     2415374.538      576674.7352415626.74387523576226.015562059
2415587.41533309575873.384572362
#Sta/Elev= 30
       0  2301.3    38.9  2282.8      53 2276.93   111.8 2261.51  132.012257.001
  230.792233.735  291.392216.613   332.6 2205.12   344.4 2202.99  354.842199.922
   360.4 2198.22   381.2 2189.22   405.7 2184.85   410.9 2184.76   413.8 2184.87
   447.6 2189.03   461.3 2189.33   475.1 2192.71   484.3 2191.96   508.9 2196.39
   540.3 2195.53   560.8 2197.09   612.8 2196.85   640.9  2198.4  681.772197.444
   717.4 2198.33   741.8 2201.61   777.8 2203.46     814 2208.65   869.6 2213.32
#Mann= 8 ,-1 , 0
       0      .1       0  132.01     .05       0  230.79      .1       0
  291.39     .05       0  354.84      .1       0   405.7    .045       0
   413.8      .1       0  681.77     .05       0
Bank Sta=405.7,413.8
XS Rating Curve= 0 ,0
Exp/Cntr=0.3,0.1

Type RM Length L Ch R = 1 ,6002    ,73.4,72.3,71.3
XS GIS Cut Line= 3
2415449.52369675576698.2806440732415694.98555966576260.177825476
2415660.80732558575943.252382235
#Sta/Elev= 30
       0 2285.04   26.892276.607    83.4 2263.85   139.2 2247.86   176.2  2240.4
   226.7 2226.75   313.8 2197.13   324.4 2194.76     342  2186.6   350.8    2185
   373.4 2183.86   383.1 2181.37   394.9 2180.67   400.9 2180.27   406.6 2180.74
   414.6 2184.37   419.2 2185.32   433.1  2184.2   459.5 2188.65   483.4 2187.95
  498.242189.145  518.252191.259   529.9 2192.03   579.6 2190.31  615.89 2191.61
   670.7  2195.1   710.3 2193.54   763.3 2194.49   799.5 2202.72   820.9 2205.63
#Mann= 7 ,-1 , 0
       0      .1       0   26.89     .05       0   394.9    .045       0
   406.6      .1       0  498.24     .05       0  518.25      .1       0
  615.89     .05       0
Bank Sta=394.9,406.6
XS Rating Curve= 0 ,0
Exp/Cntr(USF)=0,0
Exp/Cntr=0.3,0.1

Type RM Length L Ch R = 1 ,5930    ,133.7,130.5,126.7
XS GIS Cut Line= 3
     2415519.436      576759.7752415751.18371838576287.536383394
 2415715.7763646575955.160393697
#Sta/Elev= 30
       0 2289.57   158.6 2250.74   232.12227.264   324.4 2195.19   349.2 2188.92
   377.9 2187.43   382.3 2185.87   391.2 2179.16   398.42176.948   404.6 2176.56
   413.92176.986  433.492179.467   449.1 2178.12   462.5 2183.72  470.132184.775
   480.3 2184.54   493.7 2180.86     497 2180.78   508.9 2184.58   517.9 2184.94
     529  2186.9  577.82 2185.77   617.5 2187.52  675.46 2192.43   693.9 2193.02
   722.1 2190.46   746.2 2191.47   788.6 2191.03   822.6  2195.6   860.3 2204.36
#Mann= 8 ,-1 , 0
       0      .1       0   232.1     .05       0   398.4    .045       0
   413.9     .05       0  433.49      .1       0  470.13     .05       0
  577.82      .1       0  675.46     .05       0
Bank Sta=398.4,413.9
XS Rating Curve= 0 ,0
Exp/Cntr=0.3,0.1

Type RM Length L Ch R = 1 ,5799    ,152.6,154,155.3
XS GIS Cut Line= 4
2415623.77662342576798.852479686  2415815.155706576441.321174997
 2415837.5959607576317.0366874522415823.38840935575985.233653124
#Sta/Elev= 30
       0 2283.19   62.31 2267.67    90.22260.133   147.3 2242.62   189.7    2226
   256.7  2197.3   302.1 2181.47   338.4 2178.11   366.3    2177   405.5 2177.06
  425.052178.467   434.8 2177.09   451.72170.702   459.2 2169.86   466.92170.565
   475.4 2172.05   487.6 2178.17   499.8 2179.96   516.1 2180.33   524.2 2181.82
   548.3 2179.23   576.3 2178.54  626.552185.335   640.4 2186.93   668.4  2187.6
   712.4  2185.5   740.5 2186.98   764.5 2184.32   776.5 2184.39   863.9 2191.85
#Mann= 7 ,-1 , 0
       0     .05       0   62.31      .1       0    90.2     .05       0
  425.05      .1       0   451.7    .045       0   466.9      .1       0
  626.55     .05       0
Bank Sta=451.7,466.9
XS Rating Curve= 0 ,0
Exp/Cntr=0.3,0.1

Type RM Length L Ch R = 1 ,5645    ,167.3,179.1,190.8
XS GIS Cut Line= 3
     2415716.787       576818.542415932.77766405576560.400528174
     2416087.786      576041.978
#Sta/Elev= 30
       0 2271.75    56.9 2253.82   137.9 2221.51   200.8  2203.2   220.4 2196.04
     279 2183.97   306.2 2180.53   344.8 2163.52     374 2166.92  399.33 2162.82
   417.2 2162.01   461.7 2166.19   465.9 2165.93   472.42163.026   482.6 2162.97
   495.1 2163.92   507.6 2169.13   536.1 2174.49   557.7 2174.04  586.132169.162
   599.4 2168.35   624.5 2170.75   666.2 2171.03     687 2172.56   716.3  2170.7
   749.7 2172.17   791.5 2170.22   820.7  2173.1   849.9 2181.22   877.7 2185.83
#Mann= 5 ,-1 , 0
       0     .05       0  399.33      .1       0   472.4    .045       0
   482.6      .1       0  586.13     .05       0
#XS Ineff= 2 , 0
          461.96 2167.16
Permanent Ineff=
       F       F
Bank Sta=472.4,482.6
XS Rating Curve= 0 ,0
Exp/Cntr=0.3,0.1

Type RM Length L Ch R = 1 ,5466    ,125.9,120.3,112.7
XS GIS Cut Line= 4
     2415746.285      576842.8052415999.39315102576553.322439249
2416125.29153372576535.8771199962416267.78474473576158.586951319
#Sta/Elev= 30
       0 2270.34    24.3 2262.43    72.1 2243.16   113.9 2228.03   207.8 2198.92
   247.5 2188.84   302.3 2180.84   326.9 2169.08   335.4 2163.96   346.7 2159.85
   369.6 2156.51   384.5 2158.91   390.3 2158.86   414.7 2156.55   426.8 2154.03
   453.42152.616   459.1 2151.94   464.9 2152.62   475.2 2157.19   495.4 2159.56
   562.2 2161.47   627.4 2162.08   682.3 2159.19   733.2 2163.31   767.4 2160.38
   801.6 2160.48   831.6  2163.6     853 2163.77   895.7 2171.95   914.9  2172.7
#Mann= 3 ,-1 , 0
       0     .05       0   453.4    .045       0   464.9     .05       0
#XS Ineff= 2 , 0
          387.96 2159.23
Permanent Ineff=
       F       F
Bank Sta=453.4,464.9
XS Rating Curve= 0 ,0
Exp/Cntr=0.3,0.1

Type RM Length L Ch R = 1 ,5346    ,147.8,148.6,149
XS GIS Cut Line= 2
2415830.56550172576910.9987968562416554.86970142576225.113420082
#Sta/Elev= 30
       0 2257.75    53.3 2236.42   108.3 2221.69   156.5 2215.74   174.5 2212.19
   218.6 2208.58   235.1 2205.43   326.2 2173.79   351.7 2161.94   370.1 2149.92
   384.82144.874   388.5 2144.22   396.42144.861   410.8  2148.3   451.5 2149.66
     469 2155.48   486.4  2156.7   521.5 2156.65   589.3    2153   608.6 2154.27
   702.5 2154.34   724.9 2153.06   753.4 2148.87   796.9 2151.41   832.6 2149.59
   864.5 2150.31   934.6 2147.82     946 2148.58   980.9 2155.55   997.5 2157.59
#Mann= 3 ,-1 , 0
       0     .05       0   384.8    .045       0   396.4     .05       0
#XS Ineff= 2 , 0
                          419.49         2156.97
Permanent Ineff=
       F       F
Bank Sta=384.8,396.4
XS Rating Curve= 0 ,0
Exp/Cntr=0.3,0.1

Type RM Length L Ch R = 1 ,5197    ,151.4,147.4,142.9
XS GIS Cut Line= 3
     2415898.948      576999.654 2416283.9751146576693.432796856
2416606.31437677576264.120302029
#Sta/Elev= 30
       0 2242.84    28.5 2235.61    59.2 2231.03   186.9  2222.3   197.5 2220.33
   251.5 2197.93   285.7 2188.19   308.5 2178.17   334.1 2164.06   351.2 2149.98
   365.4 2140.85   411.8 2137.75   416.6 2137.57   419.5 2137.82   432.2 2142.07
   482.1 2146.64     534 2146.49   563.1 2149.49   598.1 2146.45   633.5 2146.39
   668.1 2144.46   703.2 2147.39   747.7 2144.97   813.2 2143.67   843.2 2144.93
   883.2 2143.93   913.4 2145.76   973.4 2143.63   996.3 2144.81  1028.8 2152.35
#Mann= 3 ,-1 , 0
       0     .05       0   411.8    .045       0   419.5     .05       0
#XS Ineff= 2 , 0
          378.87 2143.71
Permanent Ineff=
       F       F
Bank Sta=411.8,419.5
XS Rating Curve= 0 ,0
Exp/Cntr=0.3,0.1

Type RM Length L Ch R = 1 ,5050    ,136.6,139,139.4
XS GIS Cut Line= 3
2415975.43394787577103.445416633 2416272.9752612576925.225128818
2416635.21240629576277.288508621
#Sta/Elev= 30
       0 2240.01     128 2212.83   183.9 2203.25   225.1 2199.95   267.9 2192.31
   301.6 2184.68     333 2174.12   362.3 2161.07   385.8 2147.78   403.4 2136.01
   420.8 2131.05   425.6 2130.48   432.8 2131.08   453.1 2135.99   471.4 2133.58
   526.4 2135.49   572.2  2140.1   623.8 2142.89   676.7 2141.43   700.5 2143.69
   741.7 2139.81   764.9 2141.28   826.6 2141.05   850.1 2139.38   876.6 2141.83
     906  2140.6   966.3 2142.89  1048.7 2142.43  1067.1 2145.28  1089.2  2151.1
#Mann= 3 ,-1 , 0
       0     .05       0   420.8    .045       0   432.8     .05       0
#XS Ineff= 2 , 0
                          453.47         2136.18
Permanent Ineff=
       F       F
Bank Sta=420.8,432.8
XS Rating Curve= 0 ,0
Exp/Cntr=0.3,0.1

Type RM Length L Ch R = 1 ,4911    ,111.6,110.7,109.7
XS GIS Cut Line= 3
2416193.73195132577197.6141805282416359.68044615 576968.46896359
2416720.18866846576320.903977384
#Sta/Elev= 30
       0    2202    37.7 2204.27   106.4 2212.47   124.9 2212.56   143.7 2210.21
   175.2 2203.35   228.6  2187.6     264 2173.33   282.9 2163.18   324.1 2131.96
   331.1 2128.09     347 2127.41     379 2128.97   431.82124.335   438.5 2124.05
   447.42124.399   470.6 2130.36   488.9 2136.97   513.4 2140.38   589.6  2136.1
     631  2136.8   663.4 2134.88     689    2136   754.4 2135.35   798.6 2138.01
   827.6 2137.53   850.5  2135.5     910 2135.72   983.3 2138.15  1024.1 2144.96
#Mann= 3 ,-1 , 0
       0     .05       0   431.8    .045       0   447.4     .05       0
#XS Ineff= 2 , 0
           378.8  2129.2  465.78         2139.51
Permanent Ineff=
       F       F
Bank Sta=431.8,447.4
XS Rating Curve= 0 ,0
Exp/Cntr=0.3,0.1

Type RM Length L Ch R = 1 ,4800    ,96.8,96.6,96.4
XS GIS Cut Line= 2
  2416374.627697577216.7566428132416786.99135167576347.916012289
#Sta/Elev= 30
       0 2180.53    26.2 2183.53    71.2 2180.42    93.3 2180.83   125.3  2183.4
   146.4 2183.31   180.6  2180.9   248.6 2173.04   261.5 2169.69   283.7 2159.85
   301.4 2150.99   329.4 2134.68   354.5 2122.02   367.52119.388   376.6  2118.7
   382.52119.525   389.5 2120.28   407.6 2128.18   420.9 2132.38   458.5 2136.21
     505 2130.63   527.2 2129.49   553.7 2131.14   572.6 2130.59     691 2132.88
   731.7 2131.82   792.8 2133.12   823.8 2130.66   907.9 2133.84   961.7 2140.77
#Mann= 3 ,-1 , 0
       0     .05       0   367.5    .045       0   382.5     .05       0
#XS Ineff= 2 , 0
          335.96 2149.52
Permanent Ineff=
       F       F
Bank Sta=367.5,382.5
XS Rating Curve= 0 ,0
Exp/Cntr(USF)=0,0
Exp/Cntr=0.3,0.1

Type RM Length L Ch R = 1 ,4704    ,127.1,126.6,125.6
XS GIS Cut Line= 2
2416464.40040974577270.522295132 2416866.1584358576377.838390569
#Sta/Elev= 30
       0 2151.57    21.5 2151.75    72.4  2155.7    95.9 2156.77   177.7 2158.23
   249.8 2163.26   278.6 2162.99   291.7 2160.52   304.1 2156.09   318.1 2149.88
   334.9 2141.86   352.8 2132.18   359.1 2128.17   371.2 2118.99   375.1 2116.87
   378.5  2116.2   383.8 2115.83   389.3 2116.18   414.5 2120.96   440.5 2121.11
     454 2122.19   520.9 2124.43   594.4 2125.89   625.3 2127.67   708.4 2126.78
   770.4 2128.51   849.1 2127.34   885.4 2130.15   927.7 2131.62   978.9 2140.23
#Mann= 3 ,-1 , 0
       0     .05       0   378.5    .045       0   389.3     .05       0
#XS Ineff= 2 , 0
                          417.83         2121.23
Permanent Ineff=
       F       F
Bank Sta=378.5,389.3
XS Rating Curve= 0 ,0
Exp/Cntr=0.3,0.1

Type RM Length L Ch R = 1 ,4577    ,117.9,117.4,116.6
XS GIS Cut Line= 4
2416490.39394442577262.5084166332416698.05826562 577060.52270142
2416890.56175795 576581.908411682416891.69385243576385.442275965
#Sta/Elev= 30
       0 2149.63    70.9  2152.6     142 2149.54   199.2 2148.36   266.2 2149.82
   302.7 2147.18   310.6 2145.51   315.6 2143.29   358.7 2114.38   367.3 2112.14
     376 2111.38   382.5 2112.38   393.2 2114.57   427.7 2114.27   448.1 2116.93
   498.1 2118.11   526.8 2122.23   561.3 2120.47   587.4 2122.83   613.1 2123.13
     626 2124.09   651.8    2122   677.7 2122.92   830.9 2122.51   854.9 2124.75
   882.9 2128.49   918.9 2128.48   950.9 2129.79   974.9 2133.01    1002 2137.94
#Mann= 3 ,-1 , 0
       0     .05       0   367.3    .045       0   382.5     .05       0
#XS Ineff= 2 , 0
                          413.76         2116.69
Permanent Ineff=
       F       F
Bank Sta=367.3,382.5
XS Rating Curve= 0 ,0
Exp/Cntr=0.3,0.1

Type RM Length L Ch R = 1 ,4460    ,72.7,69.3,65.8
XS GIS Cut Line= 4
2416512.56780375577261.8892725162416816.79453124577084.514232657
2416982.62434132576589.5802936272416929.16291146576396.051334991
#Sta/Elev= 30
       0 2148.62    58.4 2148.45   167.4 2142.01   236.8 2136.08     297 2128.18
   329.4 2125.11   377.5 2123.21   381.7 2121.71   390.2 2112.22   394.4 2109.54
     407 2108.02   412.5 2107.06   417.92108.011   423.9 2110.64     445 2110.51
   461.9 2111.95   478.9 2110.43   499.8  2113.9   548.4 2116.03   647.5 2117.02
   672.8 2118.28     700 2116.97   747.4 2116.52   837.3 2119.16   859.1 2117.02
   874.1 2116.77   920.9 2122.95  1016.9 2127.48  1058.3 2131.06  1074.9 2133.93
#Mann= 3 ,-1 , 0
       0     .05       0     407    .045       0   417.9     .05       0
#XS Ineff= 2 , 0
                          459.98          2112.2
Permanent Ineff=
       F       F
Bank Sta=407,417.9
XS Rating Curve= 0 ,0
Exp/Cntr=0.5,0.3

Type RM Length L Ch R = 1 ,4390    ,57.3,57.1,56.5
XS GIS Cut Line= 5
2416529.98330643577262.787934496 2416898.2336399577109.350295552
2416905.54370439576949.2600628132417005.43394343576584.354903868
2416954.46953575576389.670866553
#Sta/Elev= 30
       0 2146.84    51.1 2144.43   111.8  2138.7   193.9 2133.07   276.4 2124.72
   398.8 2119.06   431.8 2119.09   435.8 2117.75   439.9 2115.14   451.3 2105.96
   455.9 2104.23   459.9  2104.1   465.92105.849   471.9 2107.91   523.9 2109.03
     548 2112.68   572.3 2112.65   597.3 2114.75   638.8 2114.52   676.1 2116.22
   746.6 2114.97   804.6 2115.03   879.3 2118.23   914.4 2116.02   937.1  2116.3
   945.6 2116.96   970.4 2121.97  1016.3 2123.22  1082.5 2127.66  1138.8 2134.25
#Mann= 3 ,-1 , 0
       0     .05       0   451.3    .045       0   465.9     .05       0
#XS Ineff= 2 , 0
          440.61 2108.65  492.65         2110.09
Permanent Ineff=
       F       F
Bank Sta=451.3,465.9
XS Rating Curve= 0 ,0
Exp/Cntr(USF)=0,0
Exp/Cntr=0.5,0.3

Type RM Length L Ch R = 1 ,4333    ,84.4,84.8,85.7
XS GIS Cut Line= 5
2417049.05721741577435.6305573692416956.99463404577115.329486072
2416958.91260453576958.0559061542417058.64706984576607.067307068
2416997.27201427576398.008524006
#Sta/Elev= 30
       0 2258.92   20.242250.086  118.542210.593   161.5 2191.71   186.4    2177
   215.6 2151.08   240.5 2126.76   267.6  2106.5   273.8 2104.58   290.2 2106.93
  315.152107.253   333.3 2109.23   376.1 2106.49   388.1 2102.83   392.1 2102.25
   404.1 2102.94   416.1 2106.97   452.1 2105.66   476.1 2111.31   508.8 2110.38
   533.8 2112.77   562.9 2111.55   613.4 2113.74   700.9 2111.67   745.8 2114.96
   788.3 2115.19   855.5 2113.32   903.9 2120.16   971.5 2122.25  1073.3 2132.35
#Mann= 6 ,-1 , 0
       0     .12       0   20.24      .1       0  118.54      .1       0
  315.15     .05       0   388.1    .045       0   404.1     .05       0
#XS Ineff= 2 , 0
          331.45 2109.92
Permanent Ineff=
       F       F
Bank Sta=388.1,404.1
XS Rating Curve= 0 ,0
Exp/Cntr(USF)=0,0
Exp/Cntr=0.5,0.3

Type RM Length L Ch R = 1 ,4248    ,214.1,211.4,208.1
XS GIS Cut Line= 5
2417131.52994834577406.8610000672417037.54939449577142.181072887
2417047.13924692576965.7277881012417104.67836153576599.395425121
2417047.13924692576399.926494493
#Sta/Elev= 30
       0 2237.47    82.1 2204.37   157.2 2171.88   231.8 2143.18   244.5 2136.39
   270.1 2112.17   274.2 2109.28   282.6  2105.2  302.26 2100.78  305.67 2100.59
   330.6 2101.38   355.1 2099.45   362.7 2098.79   366.7 2099.34   378.7 2103.64
   394.7 2106.33   438.8 2107.38   458.8 2106.63   479.1 2108.22  502.832107.481
   572.2 2110.24   649.1 2109.23   677.4 2112.37   715.8 2111.32   738.2 2111.96
   758.4 2110.48   819.2 2111.42     853  2117.4   918.8 2120.29    1036 2130.01
#Mann= 6 ,-1 , 0
       0      .1       0  302.26     .05       0  305.67      .1       0
   355.1    .045       0   366.7      .1       0  502.83     .05       0
#XS Ineff= 2 , 0
          318.88 2104.28
Permanent Ineff=
       F       F
Bank Sta=355.1,366.7
XS Rating Curve= 0 ,0
Exp/Cntr(USF)=0,0
Exp/Cntr=0.3,0.1

Type RM Length L Ch R = 1 ,4037    ,189.8,186.7,183.8
XS GIS Cut Line= 3
2417359.34035761577361.2294982762417238.93629561577109.575574611
2417065.27691491576406.294449595
#Sta/Elev= 30
       0  2310.4    36.3 2295.33    58.5 2284.66   111.7 2257.07   137.2 2242.99
     258 2169.76   313.1 2137.44   370.7 2099.97   383.1 2095.15  396.582094.018
   407.8 2092.57   420.2  2092.5   428.4 2091.94   432.5 2092.51   440.8  2096.9
   453.1 2098.24   469.7 2101.59   543.8  2103.7   576.7 2106.44   613.8    2108
   638.5 2107.36   671.5 2109.33   708.6 2107.75   747.2 2109.98     791 2110.61
   799.2 2111.56   819.8 2116.44     828 2117.42   885.7 2119.46  1003.4 2128.98
#Mann= 4 ,-1 , 0
       0      .1       0  396.58     .05       0   420.2    .045       0
   432.5     .05       0
Bank Sta=420.2,432.5
XS Rating Curve= 0 ,0
Exp/Cntr=0.3,0.1

Type RM Length L Ch R = 1 ,3850    ,158.9,161.4,163.5
XS GIS Cut Line= 3
2417381.22615791 577348.678524342417409.63566893576967.645758588
2417100.30565044576413.401144242
#Sta/Elev= 30
       0 2310.42    48.4 2293.54    88.5 2276.98   265.1  2197.5     285 2187.34
   313.1 2170.45   328.6 2159.99   362.1 2135.88   381.2 2123.12   399.6 2113.35
   431.5 2093.35   445.2  2087.1   452.62085.604     459 2084.78   465.82085.828
   481.9 2092.52  489.422093.768   596.5 2098.16   605.6 2098.81   614.7 2100.47
     633 2100.57   678.8 2103.43   693.5 2105.47   724.6 2113.51   738.4 2115.32
   761.3 2115.98   797.9  2114.9     885 2116.96   940.4 2120.29  1016.8  2128.4
#Mann= 4 ,-1 , 0
       0      .1       0   452.6    .045       0   465.8      .1       0
  489.42     .05       0
Bank Sta=452.6,465.8
XS Rating Curve= 0 ,0
Exp/Cntr=0.3,0.1

Type RM Length L Ch R = 1 ,3689    ,193.5,195.9,198.2
XS GIS Cut Line= 3
2417504.06045752577287.263879648 2417550.2932531576934.337446022
2417373.66743363576388.320963715
#Sta/Elev= 30
       0 2255.45    35.1 2239.54   103.7 2212.77   164.2  2183.7   192.4 2166.54
   206.7 2160.96   216.6 2158.24   236.8 2158.06   248.9 2154.17   293.3 2129.89
   313.4 2116.81   355.9  2092.9   371.1 2088.71   429.3 2087.17   437.8 2084.99
   446.42080.635   448.8 2079.62   454.6 2078.48   462.92079.715   501.3 2086.72
     526 2087.35     547 2090.54   606.1 2091.58   666.5 2090.24   719.4  2092.2
   745.9 2095.25   786.6 2106.19   816.7 2111.77   841.3 2114.38   929.8 2120.39
#Mann= 4 ,-1 , 0
       0      .1       0   446.4     .05       0   448.8    .045       0
   462.9     .05       0
Bank Sta=448.8,462.9
XS Rating Curve= 0 ,0
Exp/Cntr=0.3,0.1
